--- 16643_ras.prj (project) ---

Proj Title=16643
Current Plan=p01
Default Exp/Contr=0.3,0.1
English Units
Geom File=g01
Flow File=f01
Plan File=p01
Y Axis Title=Elevation
X Axis Title(PF)=Main Channel Distance
X Axis Title(XS)=Station
BEGIN DESCRIPTION:
RFD model 16643 exported to HEC-RAS
END DESCRIPTION:

--- 16643_ras.p01 (plan) ---

Plan Title=Plan 01
Program Version=4.10
Short Identifier=Plan 01
Geom File=g01
Flow File=f01
Subcritical Flow
Calc Critical at every XS
Secant Critical Depth

--- 16643_ras.f01 (steady flow) ---

Flow Title=Flow 01
Program Version=5.01
Number of Profiles= 6
Profile Names=10yr,25yr,50yr,100yr,100plus,500yr
River Rch & RM=16643,50,14515.42
 1227.97 1636.91 1964.74 2174.79  3175.2  3440.2
River Rch & RM=16643,50,14317.81
 1232.32 1643.22 1972.73 2184.05 3188.71 3454.18
River Rch & RM=16643,50,   14219
 1235.83 1648.25 1979.05 2191.33 3199.34 3465.05
River Rch & RM=16643,50,14021.38
 1243.29 1658.98 1992.55 2206.88 3222.05 3488.28
River Rch & RM=16643,50,13823.76
 1245.88 1662.66 1997.15 2212.14 3229.73 3496.01
River Rch & RM=16643,50,13724.95
 1248.22 1666.08  2001.5 2217.21 3237.13 3503.74
River Rch & RM=16643,50,13626.14
 1251.58 1671.19 2008.13 2225.04 3248.56 3516.09
River Rch & RM=16643,50,13428.52
 1412.38 1888.57 2271.69 2518.97  3677.7  3917.5
River Rch & RM=16643,50,13329.71
 1414.85 1892.32 2276.55 2524.71 3686.08 3926.37
River Rch & RM=16643,50, 13230.9
 1417.36  1896.1 2281.44 2530.47 3694.49 3935.23
River Rch & RM=16643,50,13132.09
 1419.45 1899.26 2285.51 2535.27 3701.49  3942.6
River Rch & RM=16643,50,13033.29
 1421.12 1901.78 2288.77  2539.1 3707.09  3948.5
River Rch & RM=16643,50,12934.48
 1423.21 1904.92 2292.84  2543.9 3714.09 3955.86
River Rch & RM=16643,50,12835.67
 1424.47 1906.81 2295.28 2546.77 3718.29 3960.28
River Rch & RM=16643,50,12736.86
  1425.3 1908.07  2296.9 2548.69 3721.09 3963.22
River Rch & RM=16643,50,12638.05
 1429.48 1914.37 2305.04 2558.27 3735.07 3977.92
River Rch & RM=16643,50,12294.86
 1433.45 1920.45 2312.97 2567.68 3748.81  3992.6
River Rch & RM=16643,50,12056.68
 1490.16 2005.43 2422.53 2696.49 3936.88 4188.79
River Rch & RM=16643,50,11678.96
 1756.55 2404.38 2937.22 3302.38 4821.48 5097.53
River Rch & RM=16643,50,11338.76
 1758.42 2407.42 2941.33 3307.39 4828.79 5105.52
River Rch & RM=16643,50,11072.97
 1766.69 2420.76 2959.25  3329.2 4860.64 5140.11
River Rch & RM=16643,50,10804.12
 1770.84 2427.44 2968.22 3340.11 4876.56 5157.37
River Rch & RM=16643,50,10337.14
 1778.67 2440.13 2985.31 3360.94 4906.97 5190.49
River Rch & RM=16643,50,10033.24
 1781.19 2444.21  2990.8 3367.62 4916.72 5201.08
River Rch & RM=16643,50,9362.315
 2348.31 3240.72  3981.1 4496.98 6565.59 6712.81
River Rch & RM=16643,50,9140.225
 2358.79 3257.22 4003.02 4523.41 6604.19 6752.24
River Rch & RM=16643,50,8858.665
 2362.02 3262.45 4010.07 4532.01 6616.73 6765.36
River Rch & RM=16643,50,8671.513
 2445.35  3390.9 4178.84  4733.8 6911.35 7059.83
River Rch & RM=16643,50,8299.586
 2447.82 3394.98 4184.39 4740.64 6921.33 7070.38
River Rch & RM=16643,50,8143.534
 2448.92 3396.79 4186.86 4743.67 6925.77 7075.07
River Rch & RM=16643,50, 7932.97
  2451.4 3400.87 4192.42 4750.51 6935.74 7085.61
River Rch & RM=16643,50,7741.143
 2455.24 3407.22 4201.05 4761.13 6951.25    7102
River Rch & RM=16643,50,7539.948
 2459.91 3414.92 4211.53 4774.02 6970.08 7121.88
River Rch & RM=16643,50, 7309.43
 2463.65 3421.14 4220.06 4784.55 6985.44 7138.24
River Rch & RM=16643,50,6993.532
 2466.07 3425.33  4225.9 4791.86 6996.12 7149.91
River Rch & RM=16643,50,6745.941
 3202.87  4501.4  5597.6 6390.91 9330.73 9294.44
River Rch & RM=16643,50,6334.468
 3207.22 4508.86    5608 6403.93 9349.74 9314.44
River Rch & RM=16643,50,6030.548
 3238.78 4561.79 5680.84 6494.36 9481.77 9450.79
River Rch & RM=16643,50,5722.718
 3240.61 4564.93  5685.2 6499.83 9489.75 9459.15
Boundary for River Rch & Prof#=16643,50,1
Up Type= 0
Dn Type= 2
Boundary for River Rch & Prof#=16643,50,2
Up Type= 0
Dn Type= 2
Boundary for River Rch & Prof#=16643,50,2
Up Type= 0
Dn Type= 2
Boundary for River Rch & Prof#=16643,50,2
Up Type= 0
Dn Type= 2
Boundary for River Rch & Prof#=16643,50,2
Up Type= 0
Dn Type= 2
Boundary for River Rch & Prof#=16643,50,2
Up Type= 0
Dn Type= 2

--- 16643_ras.g01 (geometry) ---

Geom Title=16643
Program Version=4.10

River Reach=16643,50
Reach XY= 30
886951.357201815841468.072496868886686.795984003841836.079036926
886759.716102764842006.283010767 886538.86718728842739.575704294
886708.201441306843192.174730708887227.117733018843316.397320035
887057.095510415843614.127027026 887248.11051612843773.879892658
886940.137043067844422.146313563887065.699071125844685.089947013
886716.127442081844761.809386599886423.470032189 844569.07462184
886360.339201725  844789.5813993886287.442227614845228.979449815
886602.536877592845544.691299191 886588.45389941845773.220477302
886388.160331967846658.434412084886142.255023081846845.718595151
886034.139398247847038.357267135886292.670043161847658.526446692
886463.156836519847784.675054053886544.998844359848304.976024401
886368.605588778849263.101221212886103.484724733850076.495165203
886344.847230899850326.510652113887014.788947518850494.071875836
887249.568252021850665.633198769887467.633583423851399.585692912
888354.618271986851929.471772291888528.863594911852174.263690925

Type RM Length L Ch R = 1 ,14515.42,98.809200,98.809200,98.809200
XS GIS Cut Line= 6
886874.421919647841421.471239642886945.244175518841465.722911506
886949.993952195 841468.44872882886951.733433763841469.435746495
887014.366528605841504.523400176887034.712351387841514.530229663
#Sta/Elev= 20
9910.013315.95339916.673314.70729922.486313.93969935.544 312.4979954.416311.1857
9957.861310.77299969.653310.20849981.444308.46219993.236305.988710004.74 305.705
10012.38309.993710016.21312.991810027.67 322.71910032.85325.685410039.13328.8915
10050.59332.649810053.31333.4625 10073.5340.206210084.64344.396610095.47348.2794
#Mann= 3 , 0 , 0
9910.013    0.12       09910.013    0.12       010095.47    0.12       0
#XS Ineff= 2 , 0
       0                               0
Bank Sta=9910.013,10095.47
Exp/Cntr=0.3,0.1

Type RM Length L Ch R = 1 ,14416.62,98.809300,98.809300,98.809300
XS GIS Cut Line= 6
886733.465866139841449.766618583 886863.05594625841528.550592272
886893.431544373841548.748215269886905.778884829 841557.10427058
886927.006542902 841568.11357791886981.275196288841590.488002339
#Sta/Elev= 30
9810.863320.36499824.362318.62729836.065312.97059840.187310.50729847.768306.8406
9859.471302.06029871.174298.87639878.687295.94979882.877294.64979894.579293.7019
9917.985295.68679929.688295.74199941.391294.93339955.687297.73169964.857299.0625
 9974.17298.11129976.866297.61619988.875290.05549992.231 289.01410000.93290.1079
10010.13291.962310012.97291.9976 10024.3290.547510037.82294.874610046.47298.6336
10057.29302.2616 10068.1306.848210082.12313.374710089.74318.579910096.52324.1402
#Mann= 3 , 0 , 0
9810.863    0.12       09810.863    0.12       010096.52    0.12       0
#XS Ineff= 2 , 0
       09971.314                       0
Bank Sta=9810.863,10096.52
Exp/Cntr=0.3,0.1

Type RM Length L Ch R = 1 ,14317.81,98.809300,98.809300,98.809300
XS GIS Cut Line= 6
 886740.25156255841564.847267386886764.829618214 841579.99805368
886811.488227277841606.916059496 886841.78686936841621.910016039
886876.434813177841636.355148427886942.887950242841669.810319585
#Sta/Elev= 25
9838.293317.55029855.619313.94289867.363 311.9969878.908308.88259890.452303.8103
9897.187 300.1919901.997297.39989913.542290.92179924.951285.76779936.108280.9722
9939.259280.61489947.266279.89619958.319280.42369969.154280.08089990.822 280.076
    9999278.844510002.16278.541910010.99 280.99810013.32281.858510024.49283.4697
10033.48284.922810035.65285.360610046.82292.555310057.98304.690710066.79313.7244
#Mann= 3 , 0 , 0
9838.293    0.12       09838.293    0.12       010066.79    0.12       0
#XS Ineff= 2 , 0
       0                               0
Bank Sta=9838.293,10066.79
Exp/Cntr=0.3,0.1

Type RM Length L Ch R = 1 ,   14219,98.809300,98.809300,98.809300
XS GIS Cut Line= 6
886727.173322118841641.357334951 886786.75055544841687.568912832
886811.154458094841704.383750292886830.139342928841717.139117468
886895.117506223841767.505837277886912.236563933841778.166626356
#Sta/Elev= 30
9895.965303.52599901.909  302.779918.526300.37669931.182295.97079943.837290.0191
9956.493  282.869969.149275.52349971.364 274.425 9981.38268.65989984.468267.4369
 9993.52265.607210002.11265.827710005.63265.695210017.68267.753110020.04268.4756
10023.87269.866310030.02271.3325 10036.7271.373510042.67270.906310053.03270.6754
10055.33270.477210067.98270.189110069.35270.489310080.63274.295610085.67 277.201
10093.28279.911310101.99286.399710105.94289.120410117.73295.659310126.25296.6526
#Mann= 3 , 0 , 0
9895.965  0.0565       09895.965  0.0565       010126.25  0.0565       0
#XS Ineff= 2 , 0
       0                10039.45       0
Bank Sta=9895.965,10126.25
Exp/Cntr=0.3,0.1

Type RM Length L Ch R = 1 ,14120.19,98.809200,98.809200,98.809200
XS GIS Cut Line= 6
886668.963433434841706.714737893886712.745459261841742.798635631
886776.745557975841807.468225424886801.415374835841824.361265065
886824.914663204841835.783471416886889.501720212841857.778834847
#Sta/Elev= 30
9902.233300.74999909.657299.02769916.668296.7091 9922.35293.74669931.784287.2542
9935.564285.04089948.778278.66619959.013272.72039962.245  270.73 9976.04263.2662
9989.995 255.2159990.918 254.823    9999254.012110004.02254.416310018.18256.5589
10032.34259.388610033.41259.4822 10046.5258.974710063.33257.845810072.12256.8285
10083.88255.2238   10095255.671410106.03256.946510116.79258.409810138.13263.2868
10148.65266.711810159.11278.781110164.84284.292610169.58 288.32310174.29 290.113
#Mann= 3 , 0 , 0
9902.233  0.0868       09902.233  0.0868       010174.29  0.0868       0
#XS Ineff= 2 , 0
       0                10035.36       0
Bank Sta=9902.233,10174.29
Exp/Cntr=0.3,0.1

Type RM Length L Ch R = 1 ,14021.38,98.809300,98.809300,98.809300
XS GIS Cut Line= 6
886609.215977986841850.271740795886662.307543052841852.938538983
886718.327159186841848.801170712886774.540357456 841853.55702446
 886824.16342134841860.893108217886883.718791938841873.409660477
#Sta/Elev= 26
9921.957278.70689927.783277.12479937.828268.01889947.833257.27259957.837251.4609
9967.842 246.5789977.858247.57089997.949246.764710008.06247.8762 10018.1250.6113
10031.43252.090310038.12252.6513 10058.2251.845710068.23251.938210078.27252.1988
10088.31251.544610098.42251.669910118.63 252.49210128.74254.0949   10138255.3292
10149.08256.247610157.97257.864810169.51260.369110179.73272.909910189.95286.2112
10198.86289.6049
#Mann= 3 , 0 , 0
9921.957  0.0699       09921.957  0.0699       010198.86  0.0699       0
#XS Ineff= 2 , 0
       0                10040.14       0
Bank Sta=9921.957,10198.86
Exp/Cntr=0.3,0.1

Type RM Length L Ch R = 1 ,13922.57,98.809300,98.809300,98.809300
XS GIS Cut Line= 6
886590.321578772841975.156027748 886636.50343326841972.814908856
886684.731977039841962.079124199886781.605077317841910.868016832
886813.482767341841902.818386238886872.996008261841902.392560058
#Sta/Elev= 30
9849.343 260.3069854.021260.35429864.021259.57849874.049252.8524 9884.08251.9172
9904.233253.39119914.372252.40499924.613249.62429934.994245.68979945.387244.3327
9956.216244.57649963.547244.11839967.153243.46529983.752239.45179990.357239.1544
10002.04237.494710022.21243.604310025.56244.323910036.61245.192410047.63245.4637
10058.41246.949310068.72249.503210079.03251.3157 10089.3252.059510099.32252.2042
10109.33253.327210119.34257.544910129.36268.3425 10139.4280.636610147.42283.6735
#Mann= 3 , 0 , 0
9849.343  0.0538       09849.343  0.0538       010147.42  0.0538       0
#XS Ineff= 2 , 0
       0                10038.07       0
Bank Sta=9849.343,10147.42
Exp/Cntr=0.3,0.1

Type RM Length L Ch R = 1 ,13823.76,98.809200,98.809200,98.809200
XS GIS Cut Line= 6
886580.583357463842006.477490466886708.657879216842013.301320222
886731.796565794842018.670401213886773.577911501842036.955726013
886808.269260186842047.136730451886840.583489428842053.664265215
#Sta/Elev= 27
9826.191249.34619830.611248.90129840.621243.3823 9850.63243.74389860.639244.5464
9870.648245.21799880.657 244.3979890.666240.78979900.675240.02679910.684240.2914
9920.693 241.1549930.714242.5965  9950.8242.96489960.984240.0136 9971.25236.5342
9981.713232.84529992.596 230.141    9999229.627510003.56229.398510014.47231.6824
10025.32236.445110035.74239.576210046.16244.431810052.41 247.96110056.59250.4835
10066.86257.261210092.96269.6456
#Mann= 3 , 0 , 0
9826.191  0.0604       09826.191  0.0604       010092.96  0.0604       0
#XS Ineff= 2 , 0
       0                               0
Bank Sta=9826.191,10092.96
Exp/Cntr=0.3,0.1

Type RM Length L Ch R = 1 ,13724.95,98.809300,98.809300,98.809300
XS GIS Cut Line= 6
886542.764935201 842080.94420965886679.312767373842111.921719007
886719.023732945842119.999252348886720.989034106842120.370185545
886750.813353036842126.492817447886816.328543577842143.032658182
#Sta/Elev= 30
9818.458233.47019831.004233.9871 9836.79233.30769841.258232.41829851.512231.3117
9861.767234.79639882.275234.33719892.529236.51599902.783237.50139913.037236.5563
9923.291236.4043 9927.19236.14749933.545 235.5149943.799234.91039954.053234.7764
 9964.28232.00489974.484226.47919984.689222.56099994.894222.297210005.09224.1406
 10015.3225.457810025.51225.247710035.76226.729410046.08229.099310056.39237.0872
10066.71 246.39110077.02253.494410087.33  258.9910097.65  263.4610099.02263.8523
#Mann= 3 , 0 , 0
9818.458  0.0438       09818.458  0.0438       010099.02  0.0438       0
#XS Ineff= 2 , 0
       0                               0
Bank Sta=9818.458,10099.02
Exp/Cntr=0.3,0.1

Type RM Length L Ch R = 1 ,13626.14,98.809300,98.809300,98.809300
XS GIS Cut Line= 6
886501.625051345842147.712245612886504.499650985842148.486226534
886582.441843846842173.684626315886678.279938368842209.457849067
886692.334416642 842214.44437294886775.628004131842243.759658817
#Sta/Elev= 30
9798.899230.76369823.421227.76089833.931226.9475 9844.44224.8222 9854.95224.1859
9865.459223.40919875.969225.99239886.521225.08619887.552224.65919907.869217.9909
9918.542216.43159929.216216.18129950.564214.17969961.238215.94969971.912214.9494
9982.586214.50369986.087213.86419993.215212.2473    9999211.954810003.83212.0857
10014.43213.852410025.03219.6543 10032.8223.171910035.63224.332710046.23229.2138
10056.83233.003410062.92234.467410067.43235.674910078.03239.5588 10089.3242.5174
#Mann= 3 , 0 , 0
9798.899  0.0519       09798.899  0.0519       0 10089.3  0.0519       0
#XS Ineff= 2 , 0
       0                               0
Bank Sta=9798.899,10089.3
Exp/Cntr=0.3,0.1

Type RM Length L Ch R = 1 ,13527.33,98.809300,98.809300,98.809300
XS GIS Cut Line= 6
886573.880597489842249.164158594886606.232971301842267.380971495
886630.903964623842284.599648022886664.312700919842316.225426126
886699.080997359842336.081327901886732.714409031842349.963802062
#Sta/Elev= 26
9912.893219.80889914.178219.69919925.654217.5608 9937.13214.53459945.169212.8998
9960.713210.23699963.334209.59369972.907206.61529980.682204.74249985.816203.2418
9995.039201.8267   10001201.328510009.52201.592210013.48202.437310024.31205.3696
10026.91205.562910038.43205.930910043.81206.649310049.94207.617410061.46209.0658
10066.16210.293610072.59212.233810083.45216.570310089.01218.341510094.31220.3548
10102.55222.9107
#Mann= 3 , 0 , 0
9912.893  0.0968       09912.893  0.0968       010102.55  0.0968       0
#XS Ineff= 2 , 0
       0                               0
Bank Sta=9912.893,10102.55
Exp/Cntr=0.3,0.1

Type RM Length L Ch R = 1 ,13428.52,98.809200,98.809200,98.809200
XS GIS Cut Line= 6
886554.979764854842381.349384573886591.910522406842388.158315361
886619.495309833842390.348681907 886642.24312844842391.794040979
 886670.18599292842395.815467571886710.074325693842405.994396337
#Sta/Elev= 27
9933.772208.65759933.793208.65759934.371208.62879943.972208.28829953.762207.0702
9954.138206.99829964.303200.02569971.328196.27159974.428194.77379984.459193.8087
9994.491193.3962    9999193.2938   10001193.241210004.51193.132310014.54194.9056
10021.79197.177310024.58198.066310034.68200.7656 10044.3203.032110044.79203.1368
10050.02203.089110054.99202.988510065.31203.881110075.63205.935710085.95211.4578
10087.17212.101410091.19214.2419
#Mann= 3 , 0 , 0
9933.772   0.058       09933.772   0.058       010091.19   0.058       0
#XS Ineff= 2 , 0
       0                               0
Bank Sta=9933.772,10091.19
Exp/Cntr=0.3,0.1

Type RM Length L Ch R = 1 ,13329.71,98.809300,98.809300,98.809300
XS GIS Cut Line= 6
886524.011832408842453.187914374886531.103465906842455.678370945
886565.168530016842470.329077494 886591.63581415842483.754797328
886627.945840931842501.736824912886670.531314355842518.388752062
#Sta/Elev= 29
9926.724198.14259927.771198.00419932.193197.1565 9934.24196.76479938.482 195.928
9949.367193.53959957.834191.71569960.253 191.1959971.139188.91119971.322188.8647
 9981.67186.7256 9982.34186.67229993.546185.4555    9999184.4645   10001 184.006
10003.81183.273310004.75183.090210015.91 185.69810026.34189.644110027.07 189.939
10038.23192.292110041.52193.182210049.09195.571110050.48196.072110059.83199.2436
10070.57 203.17310077.94205.6419 10081.3206.600310087.24 207.873
#Mann= 3 , 0 , 0
9926.724    0.12       09926.724    0.12       010087.24    0.12       0
#XS Ineff= 2 , 0
       0                               0
Bank Sta=9926.724,10087.24
Exp/Cntr=0.3,0.1

Type RM Length L Ch R = 1 , 13230.9,98.809300,98.809300,98.809300
XS GIS Cut Line= 5
886472.902082786842553.957220815886551.250708166842573.656618898
886553.212386093842574.046259395 886637.60415656842594.629551502
886652.452472431842597.226735288
#Sta/Elev= 28
9918.213190.90459920.376191.03289922.489190.25689930.687187.47849940.998186.2164
 9951.31185.95729961.621183.85589963.499183.13229971.932180.04859982.243176.2634
9992.555173.1657    9999172.8765   10001172.791910002.84172.692810005.02 173.129
10013.13 175.16510023.43179.508710033.72181.350310044.01  182.8310047.23183.4327
10054.31184.6652 10064.6 187.49610074.89190.651610085.19195.486910087.87 196.765
10090.02197.791610095.37200.429410102.94203.3223
#Mann= 3 , 0 , 0
9918.213  0.0625       09918.213  0.0625       010102.94  0.0625       0
#XS Ineff= 2 , 0
       0                               0
Bank Sta=9918.213,10102.94
Exp/Cntr=0.3,0.1

Type RM Length L Ch R = 1 ,13132.09,98.809200,98.809200,98.809200
XS GIS Cut Line= 6
886449.874804078842670.819286003886507.491171395842672.683524801
886537.457497847842670.665778427886539.435059744842670.367032975
886564.479097415842668.081343236886652.394808018842665.983933118
#Sta/Elev= 26
9911.319182.88149916.447182.41839926.452177.42279936.458172.25769946.463171.0495
9956.468169.29839966.473168.81859968.966168.66429976.492168.34739986.514166.2941
9996.537164.8541    9999164.7596   10001164.688810006.59164.489510016.63166.6116
10026.15169.593910026.67  169.7510036.67170.951810046.67172.054410056.68173.2221
10066.68175.763410076.68180.481710086.69186.245110096.69191.509310106.69198.2821
10114.09199.8537
#Mann= 3 , 0 , 0
9911.319  0.0459       09911.319  0.0459       010114.09  0.0459       0
#XS Ineff= 2 , 0
       0                               0
Bank Sta=9911.319,10114.09
Exp/Cntr=0.3,0.1

Type RM Length L Ch R = 1 ,13033.29,98.809300,98.809300,98.809300
XS GIS Cut Line= 6
886487.023982375842789.418496686886513.699024209842781.773486491
886535.837708852842773.407284184886579.802167159842753.436635459
886630.600936485842737.103242102886663.457010026 842728.86908643
#Sta/Elev= 28
 9934.76170.80689943.057169.93419950.798168.4933 9953.46167.76079962.509163.0669
  9963.9162.4143 9974.59 155.988 9981.67154.4017 9985.28153.73129996.316154.2916
    9999154.6396   10001155.022710005.82 156.19410007.36156.480310018.29157.9191
10029.22158.8389 10030.6159.354510034.47 160.33810039.93161.485610050.44162.5026
10060.94163.394210071.45165.108310087.83170.122810092.37171.255110096.49173.4351
10102.68176.838810112.99182.028410121.71186.5734
#Mann= 3 , 0 , 0
 9934.76    0.12       0 9934.76    0.12       010121.71    0.12       0
#XS Ineff= 2 , 0
       0                               0
Bank Sta=9934.76,10121.71
Exp/Cntr=0.3,0.1

Type RM Length L Ch R = 1 ,12934.48,98.809300,98.809300,98.809300
XS GIS Cut Line= 6
886488.955415877842886.446415336886519.770405715842879.713567046
886571.579415015842864.335161411886589.237736283842856.863126671
 886620.26753583842844.286334033886660.718034434842829.409179566
#Sta/Elev= 30
9896.236162.09299902.424158.96649903.013158.80969912.659156.33439922.895155.4365
9927.778153.69559933.233151.80789943.665 148.3059944.343148.13759954.096 145.833
9964.527146.53859974.958148.96099979.485148.72719981.822 148.5929985.525148.2867
 9996.35146.0126    9999 146.172   10001146.302510005.96146.584410007.22146.6822
10018.01149.1067 10028.8155.743110032.58159.410710034.48 161.32610039.52 166.146
10050.18175.265510060.83182.027710061.38182.308710071.49186.949910077.58188.2572
#Mann= 3 , 0 , 0
9896.236  0.0826       09896.236  0.0826       010077.58  0.0826       0
#XS Ineff= 2 , 0
       0                               0
Bank Sta=9896.236,10077.58
Exp/Cntr=0.3,0.1

Type RM Length L Ch R = 1 ,12835.67,98.809300,98.809300,98.809300
XS GIS Cut Line= 6
886459.806460395842969.855718456886516.662386779842959.729408271
886564.761787636842954.159306031886603.310722923842952.396592472
886652.235278467842949.420369516886656.356998654842948.720065595
#Sta/Elev= 29
9856.239159.25049861.515159.40649871.672158.44449881.829157.20329883.932 156.797
9891.987154.90859902.144150.70249912.301146.0395 9913.99145.83039922.383144.7909
 9932.45144.42069942.517143.56699952.584143.10659955.103142.31089962.411139.8077
9962.649139.7266 9972.66138.7542 9982.67136.7707 9992.68135.2204    9999135.5688
   10001135.670410002.69135.752610012.71141.104510022.73150.358410032.75158.3395
10042.77161.783310050.01162.107510052.82162.1857 10054.2162.2662
#Mann= 3 , 0 , 0
9856.239  0.0877       09856.239  0.0877       0 10054.2  0.0877       0
#XS Ineff= 2 , 0
       0                               0
Bank Sta=9856.239,10054.2
Exp/Cntr=0.3,0.1

Type RM Length L Ch R = 1 ,12736.86,98.809200,98.809200,98.809200
XS GIS Cut Line= 6
886494.274969044843087.090213762886636.516688903843043.895493178
 886674.57748516843030.291651792886707.679318606843015.598719077
886735.524536525843000.608649772 886746.98935362842992.874001694
#Sta/Elev= 30
9871.247 143.7339882.463143.18899892.921142.91079903.379142.73979913.837142.2507
9924.295140.08419934.753138.91439945.211138.47139955.669138.57059966.126137.5612
9987.042 127.945  9997.5126.3365   10001126.427710007.91126.793410018.33132.8587
10019.91133.415910028.91137.154910039.53139.706810046.33 139.75510050.15139.9277
10060.32141.126410071.73142.842410073.37143.018910082.67143.237610093.61143.3142
10104.85143.783310116.21143.7822 10118.9143.853710138.19 144.63510141.99144.9287
#Mann= 3 , 0 , 0
9871.247  0.1084       09871.247  0.1084       010141.99  0.1084       0
#XS Ineff= 2 , 0
       0                               0
Bank Sta=9871.247,10141.99
Exp/Cntr=0.3,0.1

Type RM Length L Ch R = 1 ,12638.05,96.236600,96.236600,96.236600
XS GIS Cut Line= 6
886600.625616215843175.103022792886666.896622463843134.076919923
886675.927198202843128.390577235886707.635287417843093.463815317
886725.862761191843067.314574318886755.750959357843007.619134605
#Sta/Elev= 29
9923.058  136.039939.964135.63479951.725135.11179961.248  134.959963.487134.5638
9975.248128.24869980.245125.1909 9987.01122.35299998.771119.3501   10001119.8406
10010.58124.894410011.67125.693810016.25128.709410025.17 131.07510029.76131.5989
10040.05132.370410043.26132.479810056.77133.654510069.16134.219310093.31134.5068
10104.49135.323710111.13136.230110115.67137.014610126.86140.660110133.47141.9924
10138.04142.573210149.23144.6566 10155.8 144.91210157.48144.8881
#Mann= 3 , 0 , 0
9923.058  0.1031       09923.058  0.1031       010157.48  0.1031       0
#XS Ineff= 2 , 0
       0                10034.36       0
Bank Sta=9923.058,10157.48
Exp/Cntr=0.3,0.1

Type RM Length L Ch R = 1 ,12541.81,47.973100,47.973100,47.973100
XS GIS Cut Line= 4
886676.978595071843310.585885526886722.890606878843238.946320295
886745.258442224843119.133928146886762.143954411843008.598912716
#Sta/Elev= 30
9879.831132.44229898.343 132.496 9913.23132.11839922.098130.05969931.764 128.072
9945.853125.79059950.297 125.169 9957.73125.38179979.108126.5663 9989.28126.7857
9999.453126.500810009.63126.4544 10019.8126.210410029.97126.746510040.14 126.276
10050.32 126.13710070.66126.381110080.84126.705410090.98127.3838 10101.1128.2576
10111.22129.746310121.33130.494710131.45131.121310141.56133.144210151.68133.6778
 10161.8136.954110171.91139.050910182.03140.343110192.14142.712410198.62143.6264
#Mann= 3 , 0 , 0
9879.831  0.0712       09879.831  0.0712       010198.62  0.0712       0
#XS Ineff= 2 , 0
       09972.108        10055.18       0
Bank Sta=9879.831,10198.62
Exp/Cntr=0.3,0.1

Type RM Length L Ch R = 1 ,12493.84,198.978400,198.978400,198.978400
XS GIS Cut Line= 3
886714.704052069843362.334246988886761.067022933843305.156589151
886814.175431853  842979.2954958
#Sta/Elev= 30
9832.533128.6395 9854.85127.47239867.724126.50859880.599125.16449893.473126.0697
9906.146 124.864  9936.7 124.4019946.832123.79419956.964124.18679967.096122.6276
9977.228119.7621 9987.36116.17539997.492114.315310007.62114.510510027.89122.0124
10048.15123.283910068.42123.859910098.81125.144610119.08126.566210139.34127.6293
10149.47127.7303 10159.6128.068410169.73129.012810179.87129.5348   10190130.4593
10200.13132.498910210.26135.163210220.39139.126810230.53144.366510236.31146.6319
#Mann= 3 , 0 , 0
9832.533  0.0655       09832.533  0.0655       010236.31  0.0655       0
#XS Ineff= 2 , 0
       0 9960.73        10055.89       0
Bank Sta=9832.533,10236.31
Exp/Cntr=0.3,0.1

Type RM Length L Ch R = 1 ,12294.86,238.184000,238.184000,238.184000
XS GIS Cut Line= 6
886891.723307275843384.110127607886922.133852864843346.752110401
 886949.17273429843291.155372882886972.191175235843227.842973407
887011.182615094843104.870713359887045.895651502843021.507886283
#Sta/Elev= 30
9823.541121.76229836.143122.77589849.432122.74589859.538 123.8029873.853123.8175
9893.904122.00599918.597120.19319950.924119.17899961.565117.99599972.206114.3824
9982.847108.95229993.488106.458510004.08106.163710010.39107.932710014.57 109.412
10025.06112.518910046.05114.227310056.54114.509910076.56114.255910088.01113.3262
 10098.5113.015710151.39117.462910168.62119.134510172.82119.711910183.53 123.019
10194.53122.226710205.57124.489510216.61124.144910218.34124.586510220.46125.8602
#Mann= 3 , 0 , 0
9823.541  0.0655       09823.541  0.0655       010220.46  0.0655       0
#XS Ineff= 2 , 0
       0                10048.61       0
Bank Sta=9823.541,10220.46
Exp/Cntr=0.3,0.1

Type RM Length L Ch R = 1 ,12056.68,377.712000,377.712000,377.712000
XS GIS Cut Line= 5
886925.901228856843414.420468322886970.888502299843393.451582747
887022.022467275843374.018015311887069.145786687843359.255805632
887481.498870649843162.794105748
#Sta/Elev= 30
9702.446123.63719748.415123.89189767.177  121.839777.875 119.9699804.019118.7607
9820.382117.21429836.949113.7285 9851.82 111.1879862.649 109.9579884.803105.5499
9962.342106.53579973.419105.65389995.573101.606110005.56100.889510017.73103.6275
 10028.8104.669710039.88 104.75510062.03106.287810084.19106.242810095.27107.3363
10106.34107.4913 10121.8 108.55910139.57 111.99410150.65109.6167 10172.8110.0198
10194.96112.618710250.34115.0752 10272.5117.767610284.55120.112610312.93 123.885
#Mann= 3 , 0 , 0
9702.446    0.04       09702.446    0.04       010312.93    0.04       0
#XS Ineff= 2 , 0
       0                10123.74       0
Bank Sta=9702.446,10312.93
Exp/Cntr=0.3,0.1

Type RM Length L Ch R = 1 ,11678.96,340.201600,340.201600,340.201600
XS GIS Cut Line= 3
886962.639841517843586.378144087886989.079738324843586.965509678
887370.884142236843596.139834904
#Sta/Elev= 30
9904.213114.98649926.578115.29789956.587 113.892 9966.59112.49579976.593106.2162
9986.596101.63059996.59995.92414 10006.695.07045 10016.696.8320810026.6198.92654
10046.61100.305410056.62102.862510076.62101.810210086.62101.847810126.64100.3714
10136.64 99.299510156.6499.6419210166.65 100.10110186.65 100.39610196.66100.9721
10206.66 102.41110216.66104.956210226.66108.336210236.67112.555710256.67120.3736
10276.68129.860210286.68  133.6610296.69134.855710306.69136.671810312.57139.9402
#Mann= 3 , 0 , 0
9904.213  0.0934       09904.213  0.0934       010312.57  0.0934       0
#XS Ineff= 2 , 0
       0                10196.97       0
Bank Sta=9904.213,10312.57
Exp/Cntr=0.3,0.1

Type RM Length L Ch R = 1 ,11338.76,265.796400,265.796400,265.796400
XS GIS Cut Line= 2
886979.860185705843755.685728946 887345.22829797843825.583893158
#Sta/Elev= 30
9733.521 115.3089748.936113.88279759.117112.65149769.298111.8215 9779.48 111.231
9789.661111.03969830.386105.64289840.568104.7073 9860.93103.17269871.112102.1816
9891.474101.59539901.656100.09659922.01998.82745  9932.297.619589942.38196.82455
9952.563  98.0939962.74498.702469972.92595.113639983.10790.807619993.28890.21807
10003.4790.6893810013.6598.9036710023.83107.393110034.01113.935210054.38126.1376
10064.56130.878610074.74133.063710084.92138.9335 10095.1144.026610105.52148.6451
#Mann= 3 , 0 , 0
9733.521  0.1182       09733.521  0.1182       010105.52  0.1182       0
#XS Ineff= 2 , 0
       0                               0
Bank Sta=9733.521,10105.52
Exp/Cntr=0.3,0.1

Type RM Length L Ch R = 1 ,11072.97,268.844500,268.844500,268.844500
XS GIS Cut Line= 6
886782.261729882843942.508642317886946.135780869843978.101758179
886995.003299127843992.468369463887049.995966465844011.926574317
887223.028320399844083.085892264887299.507230848844111.828387072
#Sta/Elev= 30
 9626.47112.24449649.658111.56039670.053109.68329700.655107.4594 9721.18105.0802
9735.881104.18819751.968103.4698 9762.23103.55359793.018101.8859 9818.64101.0263
9852.70897.737619876.93896.001219903.45395.381429919.64994.280929952.03295.09934
9984.41593.68389 9995.2191.2459610006.0692.4185710027.7196.7858710038.54101.9227
 10060.2107.217710069.47111.553210071.03111.931810092.66106.945210095.91106.9182
10103.36107.506510114.07108.887110124.77 109.74410135.48112.335910172.26  129.77
#Mann= 3 , 0 , 0
 9626.47    0.12       0 9626.47    0.12       010172.26    0.12       0
#XS Ineff= 2 , 0
       0                               0
Bank Sta=9626.47,10172.26
Exp/Cntr=0.3,0.1

Type RM Length L Ch R = 1 ,10804.12,466.982600,466.982600,466.982600
XS GIS Cut Line= 2
886818.697338262844182.584496072887295.087072122844429.700126457
#Sta/Elev= 30
9788.585108.93949837.266108.28539874.543107.20989897.073106.16089919.604105.7995
9930.869105.16439942.135102.4463  9953.496.86373 9967.5790.929139975.93188.29544
9987.19686.724089998.46183.8697710009.7383.9264110020.9988.9128610032.2691.09856
10054.4492.8089910077.3292.2804710099.8591.1382910111.1191.4098510133.65 91.2452
10167.4489.9372110178.7190.7686510201.2498.0758410206.46100.057610223.77104.6004
10235.03106.287610257.56108.922410291.36123.615610313.89129.788110325.25133.8502
#Mann= 3 , 0 , 0
9788.585   0.086       09788.585   0.086       010325.25   0.086       0
#XS Ineff= 2 , 0
       0                               0
Bank Sta=9788.585,10325.25
Exp/Cntr=0.3,0.1

Type RM Length L Ch R = 1 ,10337.14,303.901900,303.901900,303.901900
XS GIS Cut Line= 4
886825.220525304844451.466325398886884.257690308844535.240622345
887000.171722689844616.763967119887190.135953673844732.963659491
#Sta/Elev= 30
9661.352103.56939702.376102.6337 9714.61102.91559739.077101.67829764.747100.8224
9776.97299.181839789.19894.395569801.423 90.6438 9815.57  88.6859825.87487.74165
9862.55188.212939887.00288.034559899.22889.34259 9911.21 89.05999934.655 89.7126
  9958.189.197449981.54587.532739993.26884.03243 9997.9983.0895110004.9983.41471
10017.1590.2601410028.4498.7985610036.32105.732310051.88 120.544 10063.6129.5788
10075.33139.440810087.05145.008510098.77149.050410110.49151.801610128.24152.7694
#Mann= 3 , 0 , 0
9661.352   0.049       09661.352   0.049       010128.24   0.049       0
#XS Ineff= 2 , 0
       0                               0
Bank Sta=9661.352,10128.24
Exp/Cntr=0.3,0.1

Type RM Length L Ch R = 1 ,10033.24,670.922700,670.922700,670.922700
XS GIS Cut Line= 4
 886664.11299744844366.640275003886689.284788893844436.226821236
886718.491175935844564.130207831886823.872505256844822.564486347
#Sta/Elev= 30
9581.256 105.212 9600.78104.36459643.317103.59689653.951103.00589695.027 102.186
9705.284101.39239746.314100.17579766.82898.752759777.08696.99081 9798.1992.52699
9808.98991.002559841.38790.395769856.65888.389949873.78687.991259895.385 85.1386
9906.18484.064959916.98383.529779927.78384.89232 9936.1185.215469938.58285.58052
9960.18186.12554 9981.7886.140569992.57981.6622610003.3880.5364610015.56 85.5616
10024.98 93.148810035.78101.364410046.58107.613910057.38116.379110065.55 123.811
#Mann= 3 , 0 , 0
9581.256    0.04       09581.256    0.04       010065.55    0.04       0
#XS Ineff= 2 , 0
       0                               0
Bank Sta=9581.256,10065.55
Exp/Cntr=0.3,0.1

Type RM Length L Ch R = 1 ,9362.315,222.089600,222.089600,222.089600
XS GIS Cut Line= 6
885946.485763606844727.842505289886358.015701717844781.779752791
886380.646010655 844785.12445605886382.622946086844785.427346026
886418.905795305844791.805838347886811.614439084 844861.81470567
#Sta/Elev= 30
9580.769106.36059639.783104.40889649.869104.6443 9670.04102.88789680.12699.81792
9690.21194.346329700.29792.117119720.46890.17131 9760.8189.408129801.152 89.7014
9821.32387.582919831.40887.408419992.77786.5055710114.5187.7211910144.9989.50545
10155.1489.12464 10165.389.6724710195.7789.5488410246.6788.5662710287.1989.60966
10307.51 88.853510327.8289.3207610348.1493.0836410368.4597.6140610409.08 98.4878
10419.24 104.298 10429.4115.967510439.56122.788210449.72121.695310456.43124.5568
#Mann= 3 , 0 , 0
9580.769  0.0548       09580.769  0.0548       010456.43  0.0548       0
#XS Ineff= 2 , 0
       09883.763        10160.22       0
Bank Sta=9580.769,10456.43
Exp/Cntr=0.3,0.1

Type RM Length L Ch R = 1 ,9140.225,281.559800,281.559800,281.559800
XS GIS Cut Line= 6
885795.388030834844953.795436172886009.951311546844966.542918263
886202.181496862844982.203153156886318.620363552 844999.64721218
886407.530118442845019.599629189887025.582485326845108.381862368
#Sta/Elev= 30
9462.72991.883019502.41192.255639532.464 96.09539552.49996.469529572.53495.33205
9662.69394.653339682.73290.329279692.75789.426159752.90890.375979903.65488.55602
9944.06784.980469974.49880.409169984.64178.047589994.814 71.491910005.0373.38086
10015.2678.35126   10087 80.768210107.2188.0774810188.0386.5418810218.3488.07751
10339.5790.3019410390.0888.94121 10450.791.2263910501.2191.3048110521.42  92.705
10592.1392.5683210602.2493.5134510642.65106.619510662.85109.448610703.85120.8292
#Mann= 3 , 0 , 0
9462.729  0.0403       09462.729  0.0403       010703.85  0.0403       0
#XS Ineff= 2 , 0
       0                10174.94       0
Bank Sta=9462.729,10703.85
Exp/Cntr=0.3,0.1

Type RM Length L Ch R = 1 ,8858.665,187.152100,187.152100,187.152100
XS GIS Cut Line= 3
885918.986573245845358.102303786885946.688996756845347.772234917
 887018.09348739845128.015577409
#Sta/Elev= 30
9597.99289.412219625.75583.888589641.35582.488079676.87582.007899717.707 83.2778
9768.74883.114659932.07977.934529952.49675.872699972.91277.03693 9983.1274.07376
9993.32869.5596210013.7475.4050110023.9576.44011 10085.277.8320110126.0383.38023
10177.0885.9098210217.91 85.301310289.3786.1504310299.5787.46042 10330.287.65613
10371.0389.8779510411.8689.1785310432.2890.13647 10462.9  88.62310513.9590.89023
 10585.492.1013310636.4491.7215610656.86 95.107910687.49107.060410721.27115.8533
#Mann= 3 , 0 , 0
9597.992    0.04       09597.992    0.04       010721.27    0.04       0
#XS Ineff= 2 , 0
       0 9866.05        10270.55       0
Bank Sta=9597.992,10721.27
Exp/Cntr=0.3,0.1

Type RM Length L Ch R = 1 ,8671.513,371.927600,371.927600,371.927600
XS GIS Cut Line= 2
885963.018293508845618.167694819887027.929899659845142.797042229
#Sta/Elev= 30
9471.20591.112789495.27791.02515 9517.1888.387659528.13183.944269582.88680.94573
  9714.379.579589790.95780.61264 9911.4275.138169969.62375.105629977.12674.32929
9994.15668.821549999.02868.5395310009.9869.7556210031.8881.1783310053.7884.47685
10075.6984.2617810097.5985.5130910108.5484.26882 10207.185.15287 10250.988.66011
10404.2290.3786210437.07  92.79610448.0291.8725410524.6893.2154210557.5391.34204
10568.4993.5902610579.4497.5071710590.39103.850110607.46110.8703 10637.4116.2933
#Mann= 3 , 0 , 0
9471.205  0.0413       09471.205  0.0413       0 10637.4  0.0413       0
#XS Ineff= 2 , 0
       09791.362                       0
Bank Sta=9471.205,10637.4
Exp/Cntr=0.3,0.1

Type RM Length L Ch R = 1 ,8299.586,156.052100,156.052100,156.052100
XS GIS Cut Line= 2
885965.437416004845632.922038357886962.749143889845740.916220417
#Sta/Elev= 30
9368.00590.943359387.68290.898239417.85883.002459437.97583.204759458.09282.10588
9508.38483.314699578.79382.904029679.37881.330059699.49579.411569749.78777.10071
9810.13876.710959840.31377.570499850.37178.789679890.605 76.38559910.72277.23271
9950.956 76.06919981.13172.70835 9991.1965.6325410001.2563.3103810011.3167.86534
10021.3776.2020210031.4278.6376710121.9578.1811410152.1376.61535 10182.376.56608
10222.5381.1949110262.7783.04073   1030383.2690710323.1284.3640910371.1589.59045
#Mann= 3 , 0 , 0
9368.005  0.0457       09368.005  0.0457       010371.15  0.0457       0
#XS Ineff= 2 , 0
       09839.409        10041.81       0
Bank Sta=9368.005,10371.15
Exp/Cntr=0.3,0.1

Type RM Length L Ch R = 1 ,8143.534,210.563900,210.563900,210.563900
XS GIS Cut Line= 6
885802.846169486 845813.22182414886194.698111334845818.210542165
886352.491499279845826.849010583886491.237289628845841.878103582
886803.259905086845895.588104871887932.645432377 846119.71366056
#Sta/Elev= 30
9231.49192.507449273.64987.659149383.65786.867269523.66981.807779673.72483.45731
9693.74380.18995    979476.337069844.29277.6334210036.3172.5269710249.5873.90995
10361.7269.6915410382.1166.3333810453.4868.7020310484.0666.7514810524.8470.77448
 10616.672.9162410718.5570.9178510840.8972.3287710891.8669.3505310993.8172.71944
11054.9868.6400211075.3764.6899911156.9367.2092111197.7171.3117411207.9173.24977
 11218.179.4508111238.4978.4691711258.8884.8195811309.8686.7343911389.02100.4978
#Mann= 3 , 0 , 0
9231.491  0.0425       09231.491  0.0425       011389.02  0.0425       0
#XS Ineff= 2 , 0
       09857.679         10175.4       0
Bank Sta=9231.491,11389.02
Exp/Cntr=0.3,0.1

Type RM Length L Ch R = 1 , 7932.97,191.826600,191.826600,191.826600
XS GIS Cut Line= 4
885851.961531957845952.760347555886238.381740036846017.837772257
886805.396116985846101.623329874887771.289660446846296.070406853
#Sta/Elev= 30
9307.27789.708589361.06285.091049401.62584.99316 9452.3380.847869523.31582.17236
9695.70980.133639736.15475.578319756.37269.87087 9766.48 69.11999948.43569.83474
9968.65272.234399998.97862.8525410009.0963.89896 10029.370.7471910221.3770.63965
10241.5872.3887110251.6969.1572810302.5169.5463910333.11 66.710910394.3165.86477
10486.1268.7615110567.7267.5252310812.5470.7636510846.7968.4225910873.74 62.5917
10914.5562.4642111077.7572.1642211098.1677.8711111138.96  84.34211257.5892.77834
#Mann= 3 , 0 , 0
9307.277  0.0609       09307.277  0.0609       011257.58  0.0609       0
#XS Ineff= 2 , 0
       0 9865.69        10345.84       0
Bank Sta=9307.277,11257.58
Exp/Cntr=0.3,0.1

Type RM Length L Ch R = 1 ,7741.143,201.195300,201.195300,201.195300
XS GIS Cut Line= 6
885772.654322317846117.164963787885997.781542207846145.199836999
886151.848671867846171.479555565886304.317152914846203.608703665
 886706.15445117846295.978076377887513.428513905846494.193476873
#Sta/Elev= 30
9255.17584.739149338.03583.308269388.38479.657529600.974 80.50879655.42874.49761
9692.67476.059149713.11372.669359753.99171.061149846.35476.541889877.24170.14386
9969.88669.1730410000.3859.2825210010.5361.3274310020.6870.7605210030.86 74.5604
10041.1269.9725510051.3869.6987310195.1366.9561210246.5869.1593910277.47 65.9353
10287.77  61.94810308.3659.2209710370.1564.2475410401.0462.5349510504.0165.91448
10617.2759.1758210689.3560.6977110720.2569.0333710957.34 73.924711037.8384.05658
#Mann= 3 , 0 , 0
9255.175  0.0534       09255.175  0.0534       011037.83  0.0534       0
#XS Ineff= 2 , 0
       09874.049        10438.27       0
Bank Sta=9255.175,11037.83
Exp/Cntr=0.3,0.1

Type RM Length L Ch R = 1 ,7539.948,230.518000,230.518000,230.518000
XS GIS Cut Line= 6
885968.221674893846314.317257584886098.543286299846340.495903653
886342.145925839846403.345903801886411.580430473846425.868030036
886473.965496938846451.737526261887457.915816303846785.667155344
#Sta/Elev= 30
9515.88180.910139634.98778.944849676.02276.203379696.59170.913569737.72873.36546
9799.58967.830079830.73171.946549913.94671.6724910157.7563.9133310199.9765.30566
10210.5464.6844210231.6757.4884710273.2357.3996110326.7759.9254110397.0468.64756
10443.0164.9985710506.4165.1509410527.5466.4554610538.1170.4037710551.8171.50584
10601.51 68.102910686.0471.1534710728.3168.1458310812.8470.3268310833.9766.57371
 10855.169.6376410897.3764.7480410929.0766.89046 10950.265.8704711080.0889.24336
#Mann= 3 , 0 , 0
9515.881  0.0477       09515.881  0.0477       011080.08  0.0477       0
#XS Ineff= 2 , 0
       09837.859        10439.54       0
Bank Sta=9515.881,11080.08
Exp/Cntr=0.3,0.1

Type RM Length L Ch R = 1 , 7309.43,315.898300,315.898300,315.898300
XS GIS Cut Line= 6
885957.527845563846447.473088262  886142.6871965846533.014309242
886331.394387659846637.979701696886782.862414119846818.556920634
887099.822532354846902.262280917887573.582297922846979.421459536
#Sta/Elev= 30
9519.61381.191389853.21874.097849876.28371.571749898.89965.290219975.47862.27857
9996.77757.7808410007.4858.1799610018.1163.8907410028.7565.8414410114.9262.27867
10147.6363.7776510169.4457.5510910176.2557.4850210256.6760.0372210267.5863.50863
10321.7163.5840710364.6257.3541610407.15 63.190410550.4163.0569310646.6965.88712
10759.4362.6751110840.8268.9443910861.1763.7919310891.6962.47873 10932.3 64.5839
10952.5761.7996611033.56  77.507 11094.293.0758811225.57141.474111234.24141.4663
#Mann= 3 , 0 , 0
9519.613  0.0432       09519.613  0.0432       011234.24  0.0432       0
#XS Ineff= 2 , 0
       09783.896        10412.08       0
Bank Sta=9519.613,11234.24
Exp/Cntr=0.3,0.1

Type RM Length L Ch R = 1 ,6993.532,247.590800,247.590800,247.590800
XS GIS Cut Line= 2
885674.605085864846745.152328136887416.361516137847112.731481309
#Sta/Elev= 30
9520.32771.389879571.83271.682959735.35664.037479786.45765.149639857.99959.62377
 9888.6661.743329909.10159.824599919.32153.564899939.76160.790289970.42260.90726
10001.0852.9966510031.7462.6692510144.1764.0822710287.2562.3506810317.9158.07334
10471.21 57.565110491.66 54.6886 10512.158.5824910552.9854.7568810583.6462.26391
10675.6259.7366410910.69 62.640310992.4558.9844511033.3361.7368811063.9958.15033
11084.4361.3727311166.1993.1631411237.73130.2376 11268.4150.438511300.45 164.252
#Mann= 3 , 0 , 0
9520.327  0.0526       09520.327  0.0526       011300.45  0.0526       0
#XS Ineff= 2 , 0
       0 9952.31        10608.16       0
Bank Sta=9520.327,11300.45
Exp/Cntr=0.3,0.1

Type RM Length L Ch R = 1 ,6745.941,411.472400,411.472400,411.472400
XS GIS Cut Line= 6
 885872.46269367847027.312662038 886579.64565761 847161.86002799
886720.391717032847191.963304407 887011.39918404847234.080230325
887093.921278945847248.795603335887219.845196818847277.607806458
#Sta/Elev= 30
 9832.4187.238099916.44783.037269926.62880.510929987.71852.66552  9997.951.44731
10008.0852.5649510018.26 59.647910028.4460.7124110058.9954.8643410130.2660.36181
10191.35 60.687310303.3557.8538310333.8953.2310810344.08 53.705910354.26 59.5164
10415.35 61.600810506.9559.2690310537.4152.6365510588.5249.6789110609.0549.98067
10629.5756.9592410660.1658.8736910812.1659.6454310933.3355.9565110973.7258.80958
11044.7379.3301111065.0490.1195711105.92 102.895 11157.1131.673911203.31153.2708
#Mann= 3 , 0 , 0
 9832.41  0.0495       0 9832.41  0.0495       011203.31  0.0495       0
#XS Ineff= 2 , 0
       0                10674.01       0
Bank Sta=9832.41,11203.31
Exp/Cntr=0.3,0.1

Type RM Length L Ch R = 1 ,6334.468,303.920500,303.920500,303.920500
XS GIS Cut Line= 6
886019.248812024 847458.73188158886413.412693704847397.902567554
886629.797995765847397.441387547886676.231735048847394.883749496
886734.562048988 847395.65677458 886861.56161694847401.860546614
#Sta/Elev= 30
9807.514109.81859823.452106.79289843.689105.91279863.92598.396849944.87280.13071
9985.346  52.3229995.46449.76916 10015.749.6593810035.9456.7750310046.0657.25023
10096.6554.1848910106.7756.72588   1012757.4524310157.3655.13416 10177.658.38147
10217.9356.6066110307.9358.4065910327.9354.8361510347.9348.2054510377.9347.09448
10397.9348.3368410427.9455.3376810508.0155.8033510518.0157.9353310528.0160.49738
10538.0265.8803110548.0374.4469210558.04 79.4272 10608.195.5283510654.72114.9199
#Mann= 3 , 0 , 0
9807.514  0.0565       09807.514  0.0565       010654.72  0.0565       0
#XS Ineff= 2 , 0
       0                10514.38       0
Bank Sta=9807.514,10654.72
Exp/Cntr=0.3,0.1

Type RM Length L Ch R = 1 ,6030.548,307.829500,307.829500,307.829500
XS GIS Cut Line= 6
885879.525156568847808.832611779886448.664702825847676.549926327
886538.832815781847660.885340088886642.796861867 847646.46465856
886757.465286507847633.979479782886832.338939585847627.345692189
#Sta/Elev= 30
9538.82775.376949599.92772.259339688.17970.583959831.91160.14619 9924.3158.28043
9934.57656.397359965.37656.173059975.64355.247169985.909 50.725110006.4447.58045
10016.7147.2752310026.9852.3849110068.0452.1283610078.3154.4065310098.8452.66675
10139.7253.0269610149.8754.1004210180.3253.2723710200.6255.7406810220.8855.07143
10241.07 51.062110271.3548.3944210321.8352.3752310382.1955.1922610392.2558.12604
10412.3669.9607510472.6494.5324510492.72105.419410502.76106.972210510.13106.5142
#Mann= 3 , 0 , 0
9538.827  0.0534       09538.827  0.0534       010510.13  0.0534       0
#XS Ineff= 2 , 0
       0                               0
Bank Sta=9538.827,10510.13
Exp/Cntr=0.3,0.1

Type RM Length L Ch R = 1 ,5722.718,283.185200,283.185200,283.185200
XS GIS Cut Line= 6
886037.112343843847987.982077872886465.424552212847933.810867342
886528.595322863847922.558927048886591.465650742847907.787061847
886812.408778178847848.665341237886895.409824208847831.749690498
#Sta/Elev= 30
9541.06383.890049599.41282.404549639.73177.39414 9649.8175.251929700.20956.08519
9841.32455.40381 9962.2851.163639982.51447.565969992.67144.3140810002.8343.48973
10012.9945.1185510023.14 49.3131 10033.351.07234 10053.852.1440210084.6252.33788
10115.5748.0312210157.0746.5750710198.6149.5407210240.14 63.415510250.51  64.094
10271.1262.6644610281.4266.7199610291.7375.2843810302.03 80.798410312.3483.42643
10353.3381.8616110383.9482.3321810394.1585.5046510404.3690.4731210414.9889.79365
#Mann= 3 , 0 , 0
9541.063   0.056       09541.063   0.056       010414.98   0.056       0
#XS Ineff= 2 , 0
       0                               0
Bank Sta=9541.063,10414.98
Exp/Cntr=0.3,0.1

Type RM Length L Ch R = 1 ,5439.533,321.929900,321.929900,321.929900
XS GIS Cut Line= 6
886049.991157675848119.812811239 886065.53114473848121.873773767
886262.064765585848150.869249831886378.567292477  848172.9976184
886418.400450891848183.029566339 887315.39377896848324.350417489
#Sta/Elev= 30
9501.18795.057089637.62572.449299657.84267.64469 9667.9559.830679698.27551.92486
9932.48551.231039983.10146.6771310013.4740.1487510043.8441.6049610094.4649.05845
10145.0748.4997910175.4442.9019110205.8141.7242510215.9443.9106910226.0656.26003
10236.1863.5093710246.3170.2720710256.4372.5353210357.6767.0584110401.89 61.6696
10479.1559.2486410570.2669.2828210661.3771.4270110671.4973.3301710681.6180.06852
10701.8699.9743310711.98104.777810742.35 106.39910752.48110.472110783.24131.4271
#Mann= 3 , 0 , 0
9501.187    0.04       09501.187    0.04       010783.24    0.04       0
#XS Ineff= 2 , 0
       0                               0
Bank Sta=9501.187,10783.24
Exp/Cntr=0.3,0.1

Type RM Length L Ch R = 1 ,5117.603,246.904000,246.904000,246.904000
XS GIS Cut Line= 6
 885963.63719855848405.323415583886070.603754296848424.790910593
886404.814795764848499.465364003886542.775118207848527.695134272
886641.798982178 848555.99961944887304.122447249848640.353730385
#Sta/Elev= 30
9445.83280.064289528.53269.133549589.71668.104229630.60465.103999681.71353.08274
9702.20650.838389794.57749.145189804.84146.961049825.36848.739859866.42146.82122
9917.61748.092249938.02446.735299999.24637.8080410050.4242.1901810081.32 41.5521
10112.7848.25786 10154.251.2990810184.4449.8708410194.5251.4600910244.92 50.6247
10305.41 52.655910325.5751.0875910355.8152.33544 10466.7 49.894910537.2751.07741
10567.5158.29197 10728.861.4891410748.9662.6973710769.1269.8385210808.5670.99408
#Mann= 3 , 0 , 0
9445.832  0.0417       09445.832  0.0417       010808.56  0.0417       0
#XS Ineff= 2 , 0
       0                10170.64       0
Bank Sta=9445.832,10808.56
Exp/Cntr=0.3,0.1

Type RM Length L Ch R = 1 ,4870.699,246.904100,246.904100,246.904100
XS GIS Cut Line= 6
886024.164017407848682.266791898886593.146490941848786.490147155
886700.465414309 848809.18778436886951.201114121848868.588918001
887107.746852245848900.986541675888118.226686572 849129.90239238
#Sta/Elev= 30
9538.168101.88329549.19598.76645  9589.995.005999661.13474.815999732.36750.84053
9773.04646.631119884.74745.42316 9935.5242.10692 9955.8337.4490610037.1436.88108
10098.1749.0009210108.3449.1793910364.5845.3516610415.9647.2775210487.8742.50996
10620.6343.8069210661.5548.4973610743.5845.8330610835.8650.4398610928.1451.24393
11020.4246.2177511061.4350.5985311092.1951.52063 11133.246.1895811348.5346.89669
11399.7940.4629911440.8148.5292611481.82 50.9029 11574.155.3504511679.9456.44792
#Mann= 3 , 0 , 0
9538.168  0.0415       09538.168  0.0415       011679.94  0.0415       0
#XS Ineff= 2 , 0
       0                 10305.5       0
Bank Sta=9538.168,11679.94
Exp/Cntr=0.3,0.1
